--- RUSHRN2.prj (project) ---

Proj Title=RUSHRN2
Current Plan=p01
Default Exp/Contr=0,0
English Units
Geom File=g01
Flow File=f01
Plan File=p01
BEGIN DESCRIPTION:
---------- MODELED AS PART OF WVEMD CTP PROGRAM, 2023----------
Stream Name: Rush Run II
Flood Zone:  AFH
Wetzel County, WV
HEC-RAS Version: RAS 6.3
Vertical Datum: NAVD88
Projection: NAD 1983 StatePlane West Virginia S FIPS 4702 (US Feet)
Terrain: 1-meter West Virginia FEMA R3 South Central (collected 2018-2020)
Land Use: 2019 NLCD
Hydrologic Method:
WV SIR2010-5033 regression equations
Additional Model Notes:
None
END DESCRIPTION:
DSS Export Rating Curves= 0
DSS Export Rating Curve Sorted= 0
DSS Export Volume Flow Curves= 0
DXF OffsetX= 0
DXF OffsetY= 0
DXF ScaleX= 0
DXF ScaleY= 0

--- RUSHRN2.p01 (plan) ---

Plan Title=Floodplain
Program Version=6.30
Short Identifier=Floodplain
Geom File=g01
Flow File=f01
Subcritical Flow
K Sum by GR= 0
Std Step Tol= 0.01
Critical Tol= 0.01
Num of Std Step Trials= 20
Max Error Tol= 0.3
Flow Tol Ratio= 0.001
Split Flow NTrial= 30
Split Flow Tol= 0.02
Split Flow Ratio= 0.02
Log Output Level= 0
Friction Slope Method= 1
Unsteady Friction Slope Method= 2
Unsteady Bridges Friction Slope Method= 1
Parabolic Critical Depth
Global Vel Dist= 0 , 0 , 0
Global Log Level= 0
CheckData=True
Encroach Param=-1 ,0,0, 0
Mapping Interval=1HOUR
Computation Time Step Use Courant=        0
Computation Time Step Use Time Series=    0
Computation Time Step Count To Double=0
Computation Time Step Max Doubling=0
Computation Time Step Max Halving=0
Computation Time Step Residence Courant=0
Run HTab= 0
Run UNet= 0
Run Sediment= 0
Run PostProcess= 0
Run WQNet= 0
Run RASMapper= 0
UNET Theta= 0
UNET Theta Warmup= 0
UNET ZTol= 0
UNET ZSATol= 0
UNET MxIter= 0
UNET Max Iter WO Improvement= 0
UNET MaxInSteps= 0
UNET DtIC= 0
UNET DtMin= 0
UNET MaxCRTS= 0
UNET WFStab= 0
UNET SFStab= 0
UNET WFX= 1
UNET SFX= 1
UNET Gravity=32.17405
UNET 1D Methodology=Finite Difference
UNET DSS MLevel= 1
UNET Pardiso=0
UNET DZMax Abort= 0
UNET Use Existing IB Tables= 0
UNET Froude Reduction=False
UNET Froude Limit= 0
UNET Froude Power= 0
UNET D1 Cores= 0
UNET WindReference=Eulerian
UNET WindDragFormulation=Hsu (1988)
UNET D2 Coriolis=0
UNET D2 Cores= 0
UNET D2 Theta= 1
UNET D2 Theta Warmup= 1
UNET D2 Z Tol= 0.01
UNET D2 Volume Tol= 0.01
UNET D2 Max Iterations= 20
UNET D2 Equation= 0
UNET D2 RampUpFraction=0.1
UNET D2 TimeSlices= 1
UNET D2 Turbulence Formulation=Non-Conservative (original)
UNET D2 Eddy Viscosity=0.3
UNET D2 Transverse Eddy Viscosity=0.1
UNET D2 Smagorinsky Mixing=0
UNET D2 BCVolumeCheck=0
UNET D2 Cores=0
UNET D2 SolverType=PARDISO (Direct)
UNET D2 Minimum Iterations= 3
UNET D2 Maximum Iterations= 30
UNET D2 Restart Number= 10
UNET D2 Relaxation Coeff=1.3
UNET D2 SOR Precondition Iterations= 10
UNET D2 ILUT Maximum Fill= 8
UNET D2 ILUT Tolerance=1E-08
UNET D2 Convergence Tolerance=0.00001
UNET D1D2 MaxIter= 0
UNET D1D2 ZTol=0.01
UNET D1D2 QTol=0.1
UNET D1D2 MinQTol=1
Write IC File= 0
Write IC File at Fixed DateTime=0
Write IC File at Sim End=0
Echo Input=False
Echo Parameters=False
Echo Output=False
Write Detailed= 0
HDF Write Warmup=0
HDF Write Time Slices=0
HDF Flush=0
HDF Compression= 1
HDF Chunk Size= 1
HDF Spatial Parts= 1
HDF Use Max Rows=0
HDF Fixed Rows= 1
Calibration Method= 0
Calibration Iterations= 20
Calibration Max Change=0.05
Calibration Tolerance=0.2
Calibration Maximum=1.5
Calibration Minimum=0.5
Calibration Optimization Method= 1
WQ AD Non Conservative
WQ ULTIMATE=-1
WQ Max Comp Step=1HOUR
WQ Output Interval=15MIN
WQ Output Selected Increments= 0
WQ Output face flow=0
WQ Output face velocity=0
WQ Output face area=0
WQ Output face dispersion=0
WQ Output cell volume=0
WQ Output cell surface area=0
WQ Output cell continuity=0
WQ Output cumulative cell continuity=0
WQ Output face conc=0
WQ Output face dconc_dx=0
WQ Output face courant=0
WQ Output face peclet=0
WQ Output face adv mass=0
WQ Output face disp mass=0
WQ Output cell mass=0
WQ Output cell source sink temp=0
WQ Output nsm pathways=0
WQ Output nsm derived pathways=0
WQ Create Restart=0
WQ Fixed Restart=0
WQ System Summary=0
WQ Write To DSS=0
Sorting and Armoring Iterations= 10
XS Update Threshold= 0.02
Bed Roughness Predictor= 0
Hydraulics Update Threshold= 0.02
Energy Slope Method= 1
Volume Change Method= 1
Sediment Retention Method= 0
Sediment TS Multiplier= 1
Warm Up Method= 0
XS Weighting Method= 0
Number of US Weighted Cross Sections= 1
Number of DS Weighted Cross Sections= 1
Upstream XS Weight=0
Main XS Weight=1
Downstream XS Weight=0
Number of DS XS's Weighted with US Boundary= 1
Upstream Boundary Weight= 1
Weight of XSs Associated with US Boundary= 0
Number of US XS's Weighted with DS Boundary= 1
Downstream Boundary Weight= 0.5
Weight of XSs Associated with DS Boundary= 0.5
Percentile Method= 0
Sediment Output Level= 3
Mass or Volume Output= 0
Output Increment Type= 1
Profile and TS Output Increment= 1
Transport Output Increment 1
XS Output Flag= 0
XS Output Increment= 10
Read HDF5 Sediment Hotstart= 0
Sediment Hotstart Type= 0
Write Gradation File= 0
Read Gradation Hotstart= 0
Write HDF5 File= 1
Write Binary Output= 1
Write DSS Sediment File= 0
DSS Sediment Output Type= 1
SV Curve= 0
Specific Gage Flag= 0
Subcell Erosion Methods= 0
Subcell Deposition Methods= 0
Advection Scheme= 1
Matrix Solver= 0
Implicit Weighting Factor= 1
Maximum Outer Loop Convergence Iterations= 5
Convergence Maximum Absolute= 0.001
Convergence RMSE= 0.0001
Grain Fractions Max Abs Error= 0.001
Max Subgrid Regions= 1
Max Subgrid Length Scale= 3.402823E+38
Initial Layer Thickness= 3.402823E+38
Min Layer Thickness= 3.402823E+38
Max Layer Thickness= 3.402823E+38
Number of Layers= 5

--- RUSHRN2.f01 (steady flow) ---

Flow Title=Flow
Program Version=4.00
Number of Profiles=1
Profile Names=F01pct
River Rch & RM=RUSHRN2,Main,11002
     722
River Rch & RM=RUSHRN2,Main,7040
     843
River Rch & RM=RUSHRN2,Main,5997
     977
River Rch & RM=RUSHRN2,Main,3192
    1140
Boundary for River Rch & Prof#=RUSHRN2,Main      ,1
Up Type=0
Dn Type=3
Dn Slope=0.004284

--- RUSHRN2.g01 (geometry) ---

Geom Title=Geometry
Program Version=6.31

River Reach=RUSHRN2         ,Main
Reach XY= 30
1703260.70360982418718.002154416     1703174.403      418891.333
     1703220.377      419192.488     1703151.675      419237.945
     1703100.019      419445.603     1703115.515       420075.29
     1702970.362      420162.072     1702831.407      421052.106
     1702665.075      421157.484     1702486.861      421519.077
     1702026.089      421915.279     1701937.757      422069.214
     1701856.658      422616.251     1701720.802      422845.087
     1701758.575      422975.906     1701670.599      423177.688
     1701768.261      423579.636     1701689.163      423774.961
     1701745.661      423972.707     1701712.537      424201.059
     1701455.807      424587.962     1700976.438      425062.682
     1701044.852      425438.924     1700571.104      426124.585
      1700326.13      426643.295     1700382.993      426770.245
     1700321.956       427826.28     1700395.308      428056.666
     1700382.394      428313.914     1700465.415      428441.413

Type RM Length L Ch R = 1 ,11002   ,497,501.6,494.4
XS GIS Cut Line= 6
1702869.81492859418861.0940062551703124.69794901418886.197958678
  1703224.264679  418895.67366151703299.02601242 418902.42069526
 1703385.8135685418919.6880491671703480.70248634418956.340206832
#Sta/Elev= 30
       0 1275.29    46.5 1254.65    82.7 1241.11   110.8 1233.86     143 1218.86
   154.8 1214.28   159.1 1211.27   167.1 1204.08   171.1 1201.83   203.3 1187.77
   230.6 1177.39   255.5 1165.34   287.7 1146.59   295.7 1137.35   297.3 1136.77
   303.7 1135.73   319.8 1136.74   448.6 1138.17   464.5 1139.98   473.1 1142.38
   491.8 1150.83   509.8 1160.26     522 1168.16   526.4 1169.97     535 1171.01
   547.9 1170.79   552.2 1171.69   568.5 1181.65   590.8  1191.5   621.4 1207.23
#Mann= 5 ,-1,0
       0      .1       0   297.3    .045       0   319.8     .05       0
  416.13     .06       0  619.69      .1       0
Bank Sta=297.3,319.8
XS Rating Curve= 0 ,0
Exp/Cntr(USF)=0,0
Exp/Cntr=0.3,0.1

Type RM Length L Ch R = 1 ,10500   ,185.9,187.5,181.8
BEGIN DESCRIPTION:
Structure 11 XS 4
END DESCRIPTION:
XS GIS Cut Line= 6
1702835.96230601419266.4081562611703017.13648434419295.185001582
1703092.41258051 419306.363456921703192.05411351419316.452347502
1703263.34301293419343.9608226721703439.89154434 419417.10601759
#Sta/Elev= 30
       0 1243.67    48.8 1227.14    56.9 1222.28      65 1215.55    73.1 1213.08
    81.2 1207.35    89.3 1203.02   125.7 1186.38   145.3  1179.2   158.1 1173.16
   166.2 1171.32   190.5  1161.7     235 1149.42   267.3 1136.16   295.4  1133.7
  305.431131.495   311.5  1130.9   323.3 1131.48   398.3 1132.58   409.3 1134.15
   424.1 1138.29     431  1141.8   445.6 1152.98   480.3 1174.83   486.1 1177.15
     502  1177.6   506.3 1179.02   550.3 1205.72   588.5 1226.75   627.2 1239.84
#Mann= 5 ,-1,0
       0      .1       0  305.43    .045       0   323.3      .1       0
  349.55     .06       0  568.48      .1       0
Bank Sta=305.43,323.3
XS Rating Curve= 0 ,0
Exp/Cntr(USF)=0,0
Exp/Cntr=0.3,0.1

Type RM Length L Ch R = 1 ,10313   ,41.9,40.8,40
BEGIN DESCRIPTION:
Structure 11 XS 3
END DESCRIPTION:
XS GIS Cut Line= 6
 1702894.4091552 419406.48674738 1703034.6930286419500.993777886
1703073.08650975419484.0120458421703090.06824179419477.367020259
1703139.53676557419476.6286840841703393.52441006419524.620535512
#Sta/Elev= 30
       0 1193.53    10.8 1189.65    40.6 1180.68    54.6 1175.54   109.3 1152.35
   138.1 1144.29   151.6 1141.79     171 1137.04   227.3 1133.67   231.4 1132.84
  237.711130.145   243.4 1128.65   246.8 1128.62   255.4 1130.11     312  1132.1
   336.4 1134.38   340.5 1136.24   371.7 1154.35   385.3 1159.37   397.5 1167.65
   405.6 1174.87   409.7 1177.02     426 1177.62   429.9 1179.08   434.1 1182.79
   450.4 1190.15     487  1212.2   503.3 1221.22   515.5 1226.69   537.3  1233.9
#Mann= 7 ,-1,0
       0      .1       0  237.71    .045       0   255.4      .1       0
  328.84     .06       0  408.84      .1       0  428.84     .06       0
  528.84      .1       0
Bank Sta=237.71,255.4
XS Rating Curve= 0 ,0
Exp/Cntr(USF)=0,0
Exp/Cntr=0.3,0.1

Type RM Length L Ch R = 1 ,10272   ,269.8,272,272.1
BEGIN DESCRIPTION:
Structure 11 XS 2
END DESCRIPTION:
XS GIS Cut Line= 6
 1702875.9507508419442.6652199951703038.38470948419545.293948436
1703058.31978623419530.5272249191703078.25486298419520.190518457
1703130.67673146419515.7605014021703388.35605682419565.229025183
#Sta/Elev= 30
       0 1192.69      57 1172.85      74 1164.49    85.4 1155.69    90.1 1153.36
   113.7 1151.08   123.2 1143.62   129.1 1140.58   245.3 1133.13   249.3 1132.68
  255.091129.376   261.3 1127.28   269.4 1127.39   277.4 1129.31   292.8 1131.15
   330.1 1131.74   342.4 1135.32   358.6 1136.48   362.7  1137.8   374.9 1147.36
   383.1 1150.72   408.8 1165.37   423.8 1176.03   444.2 1177.87   452.3 1182.72
   460.5 1184.26   484.9 1200.87   513.4 1217.54   529.7 1225.47   554.4 1234.49
#Mann= 5 ,-1,0
       0      .1       0  255.09    .045       0   277.4      .1       0
  452.01     .06       0  552.01      .1       0
Bank Sta=255.09,277.4
XS Rating Curve= 0 ,0
Exp/Cntr(USF)=0,0
Exp/Cntr=0.3,0.1

Type RM Length L Ch R = 1 ,10000   ,505.7,513.6,515.4
BEGIN DESCRIPTION:
Structure 11 XS 1
END DESCRIPTION:
XS GIS Cut Line= 6
 1702824.8563571419751.1033810821702919.34206051419750.479694679
1703179.71063426419783.8625019191703254.10188967419793.398900166
1703340.89141425419804.5278149251703433.78492926419817.193472013
#Sta/Elev= 30
       0  1199.8    51.3 1181.24    91.3 1164.69   107.4 1157.67   123.5 1145.89
   135.6 1142.43   147.7 1135.24   151.7 1133.73   216.2 1127.44   292.9 1126.89
  299.021125.688     305 1124.35     313 1125.66   333.2 1143.47   341.3 1147.67
   365.5 1157.32   377.6 1164.78   381.6 1166.43   389.7 1167.68   401.8 1167.95
   405.8 1169.32     426 1180.45   454.5 1192.06   497.4  1212.4   526.8 1228.46
   538.9 1229.86     556  1235.4   571.2 1242.04   591.4 1247.44   613.2 1258.51
#Mann= 5 ,-1,0
       0      .1       0  299.02    .045       0     313      .1       0
  366.99     .06       0  461.99      .1       0
Bank Sta=299.02,313
XS Rating Curve= 0 ,0
Exp/Cntr(USF)=0,0
Exp/Cntr=0.3,0.1

Type RM Length L Ch R = 1 ,9487    ,443.2,440.1,436.4
XS GIS Cut Line= 6
1702698.49702975420015.4220781771702932.47392401420120.142341167
1703017.85597108420193.0637832581703078.10519442420264.014756843
1703150.75596775420335.4089710121703233.26006784420401.477736503
#Sta/Elev= 30
       0  1261.5    54.1 1237.81    75.9 1235.99    80.3 1234.41   110.9 1219.05
   137.1 1202.07   220.6  1163.4   238.3 1156.13   263.1 1148.86   271.7 1145.35
   282.2 1138.24   292.7  1125.4  299.841119.042   303.2 1117.86   308.5 1117.69
   318.6    1119   329.5 1120.07   464.5 1123.12   477.7 1125.12     487 1129.19
   509.4 1129.89     515 1133.05   520.6  1139.7   526.2 1144.19   568.2  1158.3
   585.3 1165.45     623 1183.39   637.1 1187.88   647.3 1189.66   669.3 1199.32
#Mann= 5 ,-1,0
       0      .1       0  299.84    .045       0   318.6      .1       0
  471.72     .06       0  603.58      .1       0
Bank Sta=299.84,318.6
XS Rating Curve= 0 ,0
Exp/Cntr(USF)=0,0
Exp/Cntr=0.3,0.1

Type RM Length L Ch R = 1 ,9046    ,193.1,193.9,193.3
BEGIN DESCRIPTION:
Structure 10 XS 4
END DESCRIPTION:
XS GIS Cut Line= 3
1702718.23462776420510.0428371531703015.85878787  420623.5613157
1703210.92955251420639.472820996
#Sta/Elev= 30
       0 1182.37    14.9 1175.39    23.4 1170.69    49.1 1154.36    70.5 1139.13
     109 1118.87   113.3  1117.9   121.9 1117.14   198.6 1114.65   207.5 1113.84
   214.1 1114.63   224.6 1115.59   253.9  1115.3     306 1116.88   314.5 1118.13
   330.8 1123.47   346.9 1123.79   350.9 1125.66   358.9 1133.83   362.9 1137.22
   367.9 1140.35   379.1 1146.57   399.1 1158.85   423.1 1170.86   459.3 1188.38
   463.3 1189.78   475.3 1191.64   483.3 1195.85   495.4 1200.75   514.3 1207.21
#Mann= 4 ,-1,0
       0      .1       0   198.6    .045       0   214.1     .06       0
  388.54      .1       0
Bank Sta=198.6,214.1
XS Rating Curve= 0 ,0
Exp/Cntr(USF)=0,0
Exp/Cntr=0.3,0.1

Type RM Length L Ch R = 1 ,8853    ,26.2,26,25.8
BEGIN DESCRIPTION:
Structure 10 XS 3
END DESCRIPTION:
XS GIS Cut Line= 6
1702571.26227623420781.3533548451702745.11608054420722.684423977
1702796.78779947420736.1406007821702846.30653011420760.899966102
1702889.90454296420779.2003665561703100.89739525420983.734253984
#Sta/Elev= 30
       0 1166.32    26.2 1155.22    38.9 1152.48    47.3 1147.11    55.8  1140.2
      60 1137.93    68.4 1135.45    76.9 1131.78    85.3 1130.77      98 1126.88
   108.6 1124.72   114.9 1123.72   144.4 1122.67   211.4 1116.49   289.8 1114.04
   302.9 1111.68   307.2 1110.46   311.6 1110.37   315.9 1111.68   323.9 1114.01
   341.4 1115.38   361.8 1115.16   381.6 1116.53   444.9 1118.56   497.6 1121.89
   542.9 1123.27   565.6 1124.82   582.5 1127.35   599.5 1132.84   633.4 1149.56
#Mann= 5 ,-1,0
       0      .1       0   302.9    .045       0   315.9      .1       0
  339.53     .06       0  479.53      .1       0
Bank Sta=302.9,315.9
XS Rating Curve= 0 ,0
Exp/Cntr(USF)=0,0
Exp/Cntr=0.3,0.1

Type RM Length L Ch R = 1 ,8827    ,37.4,37.1,36.3
BEGIN DESCRIPTION:
Structure 10 XS 2
END DESCRIPTION:
XS GIS Cut Line= 6
1702575.56825281420801.2684965161702740.81010396420743.676059792
1702789.25234046420756.5939895251702837.15632988420785.659331422
1702881.83083688420802.883237732 1703082.5969948420997.190430789
#Sta/Elev= 30
       0 1169.12    34.5 1156.37    48.1 1149.19    75.1 1133.47    89.5 1131.35
   102.2 1126.86   107.8 1125.56   123.5 1123.37   144.6 1122.59   178.4 1119.81
   215.7 1115.59   284.3 1113.21   292.9 1111.47   297.2 1110.32   301.5 1110.14
  306.471111.491   314.3  1113.5   327.2 1114.49   354.5 1114.34   417.7 1116.91
   463.7 1120.63   490.2 1121.79   512.9 1122.02   532.7 1123.38   546.8 1125.75
   555.7 1128.26   569.4 1134.33   583.6 1138.59   597.7 1145.98   608.4 1150.57
#Mann= 5 ,-1,0
       0      .1       0   292.9    .045       0  306.47      .1       0
  339.04     .06       0  479.04      .1       0
Bank Sta=292.9,306.47
XS Rating Curve= 0 ,0
Exp/Cntr(USF)=0,0
Exp/Cntr=0.3,0.1

Type RM Length L Ch R = 1 ,8789    ,37.6,37,35.3
BEGIN DESCRIPTION:
Structure 9 XS 4 AND Structure 10 XS 1
END DESCRIPTION:
XS GIS Cut Line= 4
1702603.02763473420800.1621480361702725.62835673420795.377729617
1702902.65183825 420843.221913811703056.94933227420994.529146323
#Sta/Elev= 30
       0 1159.85    17.1  1151.2    37.1 1142.83    41.1 1140.51    45.1 1137.36
    49.1 1135.33    65.1 1133.74    81.1    1128    97.2 1123.27   104.7 1122.18
   125.3  1120.8   133.6 1119.35     146  1116.2   166.7 1114.05     233 1112.28
  239.051110.679   241.3 1109.82   249.5  1110.7   278.6 1113.85   295.2 1113.72
   330.8 1115.23   358.5  1118.5   369.7 1118.45   414.6 1120.26   467.9  1123.3
   477.7 1125.28   483.4  1127.1   490.8 1130.08   498.6  1134.4   522.2 1142.74
#Mann= 5 ,-1,0
       0      .1       0  239.05    .045       0   249.5      .1       0
  292.69     .06       0  426.07      .1       0
Bank Sta=239.05,249.5
XS Rating Curve= 0 ,0
Exp/Cntr(USF)=0,0
Exp/Cntr=0.3,0.1

Type RM Length L Ch R = 1 ,8753    ,37.4,37.1,37.5
BEGIN DESCRIPTION:
Structure 9 XS 3
END DESCRIPTION:
XS GIS Cut Line= 4
 1702595.2529548420810.329037177 1702693.9315847420858.173221371
1702893.08300141   420865.3498491703044.39023392421004.696035464
#Sta/Elev= 30
       0 1163.52    17.3 1157.29      41 1149.78    54.3 1143.36    58.7 1142.19
    68.2  1140.9    83.1 1132.45    98.8 1126.12   115.9 1116.91   123.9 1114.41
   131.9 1113.25   156.6 1112.29   243.9 1112.08   247.9 1111.74   253.1 1110.34
   255.9 1109.28   259.9 1108.98   263.1 1110.45     268 1112.18   287.9  1113.5
     304 1113.78   319.6 1116.21   401.1 1120.34   432.7 1120.58   463.4 1123.46
   470.8 1124.94     479 1127.68   487.1 1131.36     503 1139.78   514.6 1144.59
#Mann= 5 ,-1,0
       0      .1       0   253.1    .045       0   263.1      .1       0
  308.95     .06       0  438.95      .1       0
Bank Sta=253.1,263.1
XS Rating Curve= 0 ,0
Exp/Cntr(USF)=0,0
Exp/Cntr=0.3,0.1

Type RM Length L Ch R = 1 ,8715    ,209.7,215.7,218.8
BEGIN DESCRIPTION:
Structure 9 XS 2
END DESCRIPTION:
XS GIS Cut Line= 4
1702585.08606566 420843.221913811702690.34327089420896.448568726
1702885.90637378420901.8310394481703027.64476945421035.196702888
#Sta/Elev= 30
       0 1170.05    11.8 1165.11    30.3 1158.93    34.8 1156.76    43.7 1150.07
    53.8 1148.88    57.2 1147.81    75.1 1136.07    98.5 1124.21   115.5 1113.38
   119.7 1111.94   131.7 1110.52   143.7 1111.13   163.7 1110.86   231.8  1111.9
   259.8 1110.75   267.7 1108.66   271.8 1108.81  279.151110.683   295.8 1113.22
   311.8 1113.42   316.6 1114.73   327.6 1116.27   381.7 1118.45   416.8 1118.58
   450.1 1122.31   455.7 1124.15   469.9 1131.26   492.5 1144.39   508.2 1152.48
#Mann= 5 ,-1,0
       0      .1       0  217.95     .06       0   259.8    .045       0
  279.15     .06       0  423.59      .1       0
Bank Sta=259.8,279.15
XS Rating Curve= 0 ,0
Exp/Cntr(USF)=0,0
Exp/Cntr=0.3,0.1

Type RM Length L Ch R = 1 ,8500    ,501.4,502.1,499.3
BEGIN DESCRIPTION:
Structure 9 XS 1
END DESCRIPTION:
XS GIS Cut Line= 6
1702532.14335984420887.6814884991702622.54869084420949.672834337
1702702.32149717 421015.62972343 1702764.6691415421072.220489502
 1702843.3740366421133.9470720891703048.37329851 421287.69774884
#Sta/Elev= 30
       0 1191.86     9.7 1191.34    43.6 1175.27      61 1168.65    72.7 1160.38
    87.3 1156.39      97 1150.93     107  1142.8     122 1133.73   170.6 1110.83
   268.8  1108.4   317.1 1108.81   345.6 1107.35   354.1 1106.36  358.391107.393
   365.5 1112.47   371.2 1114.84   393.2 1116.59   399.7 1121.27   408.3 1124.84
   431.2 1137.59   442.6 1147.61   463.3 1157.75   508.3 1182.86   523.3 1189.29
     555 1198.71   588.3  1216.8   613.3 1233.01     634 1242.35   653.6 1246.88
#Mann= 5 ,-1,0
       0      .1       0  307.33     .06       0   345.6    .045       0
  358.39     .06       0  457.35      .1       0
Bank Sta=345.6,358.39
XS Rating Curve= 0 ,0
Exp/Cntr(USF)=0,0
Exp/Cntr=0.3,0.1

Type RM Length L Ch R = 1 ,7998    ,496.6,500,501.1
XS GIS Cut Line= 6
1702247.27024193421304.0654982631702329.14967135421350.987648502
1702560.61705618 421474.797768341702626.75143833421510.171385258
 1702705.3464255421548.7507044231702790.19730568421588.886122838
#Sta/Elev= 30
       0 1257.24      24 1250.48    37.9 1244.02    70.1 1224.78   111.3 1203.24
     125 1200.43   165.8  1178.8   186.4 1166.89   206.6 1156.68   224.7 1144.82
     252 1134.17     261 1132.08   272.1 1125.12   297.3 1102.44   306.4 1100.97
   312.4 1102.32   319.4 1103.57   363.7 1103.33   419.9  1105.5   437.8 1107.63
   451.2 1112.71   464.6 1124.26     469 1125.53   486.9 1126.66   495.8 1132.89
   513.6 1142.24   537.6 1157.26   584.4 1182.22   599.4 1189.48   613.3 1194.75
#Mann= 5 ,-1,0
       0      .1       0   297.3    .045       0   312.4      .1       0
  396.87     .06       0  501.87      .1       0
Bank Sta=297.3,312.4
XS Rating Curve= 0 ,0
Exp/Cntr(USF)=0,0
Exp/Cntr=0.3,0.1

Type RM Length L Ch R = 1 ,7498    ,259.2,253.3,252.7
BEGIN DESCRIPTION:
Structure 8 XS 4
END DESCRIPTION:
XS GIS Cut Line= 6
 1701957.1120296421583.8903979211702022.85336792 421650.72687842
  1702084.211841421713.1079872551702136.80523975421766.577368513
1702320.88065901421953.7200388461702386.62199734422020.556519344
#Sta/Elev= 30
       0 1243.39     6.5 1238.84    17.7 1228.77    38.5 1215.98    70.5 1199.48
    79.5 1195.96    90.7  1193.1   107.2 1183.87   197.7 1143.32   248.7 1126.82
     259 1121.43   268.5 1114.94   283.8 1100.56   288.3  1098.7   299.6 1097.31
   310.9  1096.4     318 1097.34   323.7 1098.23   418.4 1100.51   432.1 1102.82
   443.5 1107.11   455.1 1114.34   466.5 1115.86   494.8 1132.75   506.2 1134.83
   523.4 1135.36   533.9 1142.17   542.8 1151.75   548.5 1155.89   612.5 1186.31
#Mann= 5 ,-1,0
       0      .1       0   299.6    .045       0     318      .1       0
  396.25     .06       0  538.75      .1       0
Bank Sta=299.6,318
XS Rating Curve= 0 ,0
Exp/Cntr(USF)=0,0
Exp/Cntr=0.3,0.1

Type RM Length L Ch R = 1 ,7244    ,37.3,38.3,36.4
BEGIN DESCRIPTION:
Structure 8 XS 3
END DESCRIPTION:
XS GIS Cut Line= 4
 1701910.8551099421908.6223655891701952.05426852421963.111575366
1702012.52400132421974.4081188561702233.13885065422132.559727718
#Sta/Elev= 30
       0 1127.93    14.9 1120.92      22 1118.17    55.1  1106.7    83.3 1099.85
   91.931095.059    93.6 1094.25    96.9 1093.74     105 1095.05   117.2 1096.25
   178.5 1095.66     209 1096.17   252.4 1097.77   257.2 1100.47   271.5  1114.1
   277.3 1118.19   286.8 1123.73   298.3 1127.77   311.7  1135.5   316.3 1137.34
   321.3 1137.95   334.6 1137.99   337.5 1138.56     341 1140.62   350.8 1149.08
   370.5 1162.98   374.7  1165.4   380.5 1167.19   383.3 1168.57   401.3 1178.28
#Mann= 5 ,-1,0
       0      .1       0   91.93    .045       0     105      .1       0
  239.83     .06       0  359.83      .1       0
Bank Sta=91.93,105
XS Rating Curve= 0 ,0
Exp/Cntr(USF)=0,0
Exp/Cntr=0.3,0.1

Type RM Length L Ch R = 1 ,7206    ,164.3,166.3,167.4
BEGIN DESCRIPTION:
Structure 8 XS 2
END DESCRIPTION:
XS GIS Cut Line= 4
1701876.30097688421935.2024679191701930.79018665421994.343195603
1701993.91792969422004.3107339771702217.19078926422160.468835164
#Sta/Elev= 30
       0 1127.91    23.6 1118.32    58.8 1105.96    72.5 1100.54    85.8  1097.9
      98 1097.48   104.5 1095.32   110.1 1093.84   114.2  1093.9  119.42 1095.37
   122.3 1096.07   125.5 1096.11   166.2 1095.19     230 1095.06   242.4 1096.15
   258.1 1096.76   263.4 1099.16   266.7 1101.56   275.3 1108.95   298.3 1127.45
   312.7 1135.37   317.8 1137.19   322.7 1138.03   341.4 1138.12   344.3 1138.89
   347.1 1140.49   361.5 1154.04     373 1161.67   402.9 1177.62   416.8 1183.37
#Mann= 5 ,-1,0
       0      .1       0   104.5    .045       0  119.42      .1       0
  244.33     .06       0  394.33      .1       0
Bank Sta=104.5,119.42
XS Rating Curve= 0 ,0
Exp/Cntr(USF)=0,0
Exp/Cntr=0.3,0.1

Type RM Length L Ch R = 1 ,7040    ,83.2,79.9,76.9
BEGIN DESCRIPTION:
Structure 7 XS 4 AND Structure 8 XS 1
END DESCRIPTION:
XS GIS Cut Line= 3
1701784.59962384422022.9168056081701796.56066989422097.341092131
1702181.30765111422273.434270066
#Sta/Elev= 30
       0    1119     9.7  1115.2    38.1 1102.26    46.2 1099.48    50.3 1098.91
    74.6 1096.99    92.7  1096.4   189.1 1094.41   198.1 1093.78   215.7 1094.08
   220.1 1093.53   224.5 1092.52  231.081093.556   237.7 1094.42   255.2 1094.39
   272.8 1093.41   282.7 1094.08   285.7 1095.42   288.7 1097.89   312.4 1119.91
   321.2 1127.08     343 1139.83   347.6 1140.57   365.2 1140.62   369.6 1141.67
   387.2 1152.96   404.8 1165.19   430.5 1179.65   481.8  1204.3   498.5 1210.39
#Mann= 6 ,-1,0
       0      .1       0      40     .06       0   85.38      .1       0
   220.1    .045       0  231.08     .06       0  465.38      .1       0
Bank Sta=220.1,231.08
XS Rating Curve= 0 ,0
Exp/Cntr(USF)=0,0
Exp/Cntr=0.3,0.1

Type RM Length L Ch R = 1 ,6960    ,52.1,49.9,49.1
BEGIN DESCRIPTION:
Structure 7 XS 3
END DESCRIPTION:
XS GIS Cut Line= 6
1701655.74736727422213.8390044141701757.04816138422175.497847161
1701865.38057866422229.6373113311701907.46574069422240.712353968
 1701942.9933857422236.5254644161702145.97050821422317.444916018
#Sta/Elev= 30
       0 1126.37    13.7 1116.32    34.6 1103.86      56 1096.81    63.3 1097.74
    94.5 1097.53   197.7 1094.53   249.1 1093.73   277.9 1094.25   281.51093.167
     286  1091.7     290  1091.9     294 1093.18     298 1094.06   314.5 1094.08
   318.8  1095.6   322.2 1098.37     336 1112.88     349 1124.04   366.2 1133.88
   374.5 1139.29   380.7 1141.16   400.6 1142.41   411.2 1149.46   426.5 1158.45
   438.6 1167.48   456.6 1177.29   471.1 1184.07   508.3 1203.26   527.5 1210.26
#Mann= 5 ,-1,0
       0      .1       0      60     .06       0   281.5    .045       0
     294     .06       0     479      .1       0
Bank Sta=281.5,294
XS Rating Curve= 0 ,0
Exp/Cntr(USF)=0,0
Exp/Cntr=0.3,0.1

Type RM Length L Ch R = 1 ,6910    ,401.7,409.9,413.9
BEGIN DESCRIPTION:
Structure 7 XS 2
END DESCRIPTION:
XS GIS Cut Line= 6
 1701656.5977597  422243.12479411701739.44014942422212.905334781
1701859.58594551 422279.596513941701901.67110753422290.671556577
1701937.19875255422286.4846670251702129.54383413422361.423595603
#Sta/Elev= 30
       0 1130.39      29 1109.59    37.4  1104.4    50.1 1100.24    71.4 1097.91
    80.2 1094.68    88.5 1095.48   103.5 1095.47   123.6 1094.28   218.5 1093.18
   230.6 1092.29   271.8 1093.19   283.9 1091.67   295.1 1091.31     300 1091.56
  302.031093.174   304.1 1094.82   308.3 1101.99   312.6 1107.71   324.4 1120.03
     334 1128.65   342.6 1134.84   355.5 1141.49   359.8 1142.25   381.3 1142.41
   385.6 1144.03   389.9 1147.78   419.9  1167.4   487.1 1202.96   511.6 1213.17
#Mann= 5 ,-1,0
       0      .1       0      60     .06       0   271.8    .045       0
  302.03     .06       0  485.16      .1       0
Bank Sta=271.8,302.03
XS Rating Curve= 0 ,0
Exp/Cntr(USF)=0,0
Exp/Cntr=0.3,0.1

Type RM Length L Ch R = 1 ,6500    ,498,502.9,502.7
BEGIN DESCRIPTION:
Structure 7 XS 1
END DESCRIPTION:
XS GIS Cut Line= 6
1701549.55805467422526.6398247631701710.33726068 422617.32665126
1701779.51822467422649.4991590831701940.45819151422718.577761084
1702019.54530367422756.0681716651702102.50609575422799.965065509
#Sta/Elev= 30
       0 1170.09    44.7 1146.42    82.2 1136.11   100.2 1129.61   113.8  1122.1
   150.2 1098.23   163.9 1091.57   186.6 1088.71   252.7 1087.34   287.6  1088.4
   296.2  1090.1   300.6  1089.5   304.9  1087.2   309.3 1085.37   313.6 1084.97
   317.9 1085.23   322.3 1087.28   343.2 1104.24   348.3 1109.38   361.5 1126.09
     370 1133.62   391.8 1141.55   413.8 1142.23   425.2 1148.37   444.5 1152.79
   462.2 1167.65   484.4 1178.97   523.8 1202.82     565 1222.17   617.4 1249.52
#Mann= 5 ,-1,0
       0      .1       0   304.9    .045       0   322.3      .1       0
  401.08     .06       0  506.06      .1       0
Bank Sta=304.9,322.3
XS Rating Curve= 0 ,0
Exp/Cntr(USF)=0,0
Exp/Cntr=0.3,0.1

Type RM Length L Ch R = 1 ,5997    ,502.6,497.1,486.3
XS GIS Cut Line= 6
1701427.86702509422990.2153411661701618.50312676423037.174892917
1701684.31795576423076.881178334 1701826.1359136423180.261220917
1701911.28010026423208.6971876771702006.65458143423227.295575678
#Sta/Elev= 30
       0 1150.74    12.5  1146.7      37 1143.66    65.6 1132.21    73.8 1126.86
    90.4 1113.71   110.8 1099.95   123.2 1092.18   131.6 1088.56   160.7 1085.14
     305 1082.22   315.6 1080.25   329.2 1079.44  335.021080.375   369.4 1103.01
   389.3 1119.77   408.4 1132.46   427.5 1140.41   432.3 1141.73   455.3 1143.29
   459.5  1145.5     468 1152.02   480.6 1156.07   489.1 1159.99   505.9 1172.02
   522.8  1181.7   539.4 1189.85   566.6 1202.32   605.9 1216.11     636 1230.62
#Mann= 7 ,-1,0
       0      .1       0  303.33     .06       0   315.6    .045       0
  335.02     .06       0  383.64      .1       0  423.64     .06       0
  529.01      .1       0
Bank Sta=315.6,335.02
XS Rating Curve= 0 ,0
Exp/Cntr(USF)=0,0
Exp/Cntr=0.3,0.1

Type RM Length L Ch R = 1 ,5500    ,121.8,128.3,137.2
BEGIN DESCRIPTION:
Structure 6 XS 4
END DESCRIPTION:
XS GIS Cut Line= 6
1701446.69605568423567.4349872621701546.94224626423577.475649595
1701639.71338618423584.0048360081701717.38875575423579.836209178
 1701816.7537145 423564.831646011702070.85130343    423531.68998
#Sta/Elev= 30
       0 1136.16    45.6 1129.86    73.8 1117.03    89.9 1115.88   105.9 1109.25
     126 1098.91     146 1093.54   178.1 1079.93   214.2 1077.43   282.4 1077.33
   314.7 1074.92   322.8 1072.56   326.9 1072.64  332.341074.984     339    1079
   355.2 1083.28   371.4 1091.59   395.6  1109.8   407.7 1120.39   419.8 1127.81
     448 1139.87   472.2 1140.73   496.4  1151.6   516.6  1165.5     524 1169.13
     561 1182.37   573.1 1188.13   589.2 1198.16   601.3 1203.37   628.3  1211.5
#Mann= 5 ,-1,0
       0      .1       0   314.7    .045       0  332.34      .1       0
  361.54     .06       0  467.03      .1       0
Bank Sta=314.7,332.34
XS Rating Curve= 0 ,0
Exp/Cntr(USF)=0,0
Exp/Cntr=0.3,0.1

Type RM Length L Ch R = 1 ,5372    ,37.3,38.3,38.6
BEGIN DESCRIPTION:
Structure 6 XS 3
END DESCRIPTION:
XS GIS Cut Line= 6
1701478.53380725423698.1701107381701710.97297371423664.443643447
1701721.91128743423682.6741663071701750.16859786423710.019950597
1701839.49815988423757.4193100331702057.35290805423693.612480023
#Sta/Elev= 30
       0 1168.84    11.4 1164.25    29.9 1151.25      42 1147.46    91.1  1138.9
   110.7 1131.81   118.8 1126.25   143.1 1104.71   171.4 1087.98   187.5 1080.49
   211.1 1076.31   256.2 1075.05   264.8 1072.63   273.2 1071.29  280.91 1072.68
     287 1075.93     293 1076.77   401.4 1076.59   418.1 1077.15   430.6  1079.5
   446.1 1086.17   463.9  1096.5   509.8 1131.06   530.6  1132.1   542.9 1134.55
     559 1140.43   580.6 1150.58   600.9 1164.21     614 1168.36   623.6 1173.82
#Mann= 7 ,-1,0
       0      .1       0   264.8    .045       0  280.91      .1       0
  355.46     .05       0  466.58      .1       0  486.58     .06       0
  566.58      .1       0
Bank Sta=264.8,280.91
XS Rating Curve= 0 ,0
Exp/Cntr(USF)=0,0
Exp/Cntr=0.3,0.1

Type RM Length L Ch R = 1 ,5334    ,337.8,332.4,325.2
BEGIN DESCRIPTION:
Structure 6 XS 2
END DESCRIPTION:
XS GIS Cut Line= 6
1701478.53380725423723.6928427421701688.18482014423695.435532309
1701730.11502272423744.6579440311701779.33743444423772.915254464
1701834.02900302423800.2610387541702057.35290805423727.338947314
#Sta/Elev= 30
       0 1176.07    13.7  1170.2    29.8 1165.53      46 1155.34    58.1 1150.53
    74.2 1147.16      86 1141.93    98.5 1139.53   114.6 1133.29   134.8 1118.62
   150.9 1102.26   195.3 1080.19   217.8 1074.97   244.1 1072.34   254.7 1071.28
   260.6 1072.41   266.2 1075.25   273.2 1076.14   396.3 1075.81   442.6  1079.1
   462.2 1085.74   480.5 1095.92   505.7 1111.94   526.8 1128.45   547.8 1128.53
   556.2 1136.26   560.4  1138.3   576.4 1139.43   585.7 1141.67   629.1 1164.81
#Mann= 7 ,-1,0
       0      .1       0   244.1    .045       0   260.6      .1       0
  362.98     .05       0  474.13      .1       0  574.13     .06       0
  614.13      .1       0
Bank Sta=244.1,260.6
XS Rating Curve= 0 ,0
Exp/Cntr(USF)=0,0
Exp/Cntr=0.3,0.1

Type RM Length L Ch R = 1 ,5001    ,494.1,500,504.8
BEGIN DESCRIPTION:
Structure 6 XS 1
END DESCRIPTION:
XS GIS Cut Line= 6
1701438.54056017424019.1712885051701532.05251226424025.848112419
1701619.33022484424032.0823519231701793.88565001424044.550174758
1701955.97259617424056.1272513421702049.48454826424062.806043759
#Sta/Elev= 30
       0 1231.52    17.6 1223.95    45.7 1217.78    57.7 1212.73   101.8 1187.84
   121.9 1174.89   133.9 1165.08   145.9 1158.68     166 1152.73     178 1151.74
     186  1149.9   206.1 1142.03   214.1 1138.06   222.1 1132.64   234.8 1121.68
   242.2 1114.51   250.2    1105   254.2 1101.21   270.3 1091.53  297.651069.836
   302.3 1068.47   306.4 1068.27   310.4 1068.42   314.4 1069.74   338.4 1074.05
   350.5 1073.53   414.6 1075.91   466.9 1080.25     559 1085.11   612.5 1089.01
#Mann= 5 ,-1,0
       0      .1       0  297.65    .045       0   314.4      .1       0
  366.25     .05       0  471.25     .06       0
Bank Sta=297.65,314.4
XS Rating Curve= 0 ,0
Exp/Cntr(USF)=0,0
Exp/Cntr=0.3,0.1

Type RM Length L Ch R = 1 ,4501    ,499.5,500,499.8
XS GIS Cut Line= 6
1701290.73475343424286.2540876721701363.44326942424345.436384007
1701489.47156067424448.018527925 1701625.1934021424558.492716417
1701695.58040042424610.6267985111701771.63536642424666.267435253
#Sta/Elev= 30
       0 1242.48    28.2 1225.23    68.8 1206.81   116.3 1176.65   136.2 1159.88
   141.9  1156.5   147.6 1153.93   166.8 1149.62     176  1145.6   187.4 1142.95
   204.5 1135.94   223.6 1123.98   249.3 1105.26   269.9 1094.37   275.6 1090.22
   285.4 1081.32   295.5 1066.46     304 1064.43   314.1 1066.41   329.6  1068.4
   388.6 1069.69   414.4  1071.9   426.2 1083.45   437.7 1088.53   468.3 1098.68
   514.9  1127.1   554.2 1140.63   583.6 1149.12   596.6 1155.52   613.1 1166.07
#Mann= 5 ,-1,0
       0      .1       0   295.5    .045       0   314.1      .1       0
  376.25     .06       0  538.84      .1       0
Bank Sta=295.5,314.1
XS Rating Curve= 0 ,0
Exp/Cntr(USF)=0,0
Exp/Cntr=0.3,0.1

Type RM Length L Ch R = 1 ,4001    ,306.7,304.3,302.6
XS GIS Cut Line= 6
1700947.64521651424642.3140710891701087.92511967 424757.08811976
 1701145.9719196424804.5811350051701223.36809026424867.904499173
1701349.13621143424970.8052120061701421.69479334425030.171563089
#Sta/Elev= 30
       0 1190.79    67.8 1164.76   115.6 1143.05   129.8 1141.22   150.5 1136.48
     166 1131.48   186.7 1119.88   202.2 1108.83   217.7  1096.2     228 1091.06
   248.7 1083.52     259 1082.41     272 1082.92   279.7 1080.32   284.9 1075.22
   294.1 1063.99  296.891061.775   300.4 1060.12   305.5 1059.97   310.7 1060.25
  314.32 1061.82   319.3 1064.44     326 1065.12   433.1 1065.56   477.3 1067.94
   508.9 1067.65   538.1 1078.89   547.7 1083.72   573.3 1100.56   612.5 1131.14
#Mann= 7 ,-1,0
       0      .1       0  276.25     .06       0  296.89    .045       0
  314.32     .06       0  431.25     .07       0  588.75     .06       0
  598.75      .1       0
Bank Sta=296.89,314.32
XS Rating Curve= 0 ,0
Exp/Cntr(USF)=0,0
Exp/Cntr=0.3,0.1

Type RM Length L Ch R = 1 ,3697    ,273.7,265.5,259.9
XS GIS Cut Line= 3
1700800.48498972424964.1966308371701021.07431632 425080.87197714
1701379.30409052425152.882542437
#Sta/Elev= 30
       0 1157.11    13.2 1151.65    35.8  1145.1    58.4 1140.11    94.6 1133.97
   121.8 1122.19   153.4 1100.84   171.8 1085.61   176.1 1081.27   180.4 1073.71
   185.1 1064.22   189.6 1058.72   194.2 1056.84   198.3 1056.69   204.2 1056.89
   209.6 1058.76   213.1 1060.63   216.8 1061.57   225.8 1061.06   387.3 1061.26
   497.4 1066.59   513.8 1066.53   517.8  1067.7     526 1077.38   542.3 1090.81
   558.6 1099.69     575  1110.7   587.2 1119.87   607.6 1131.28   614.9 1133.21
#Mann= 6 ,-1,0
       0      .1       0   189.6    .045       0   209.6      .1       0
  349.55     .05       0  409.55     .06       0  549.55      .1       0
Bank Sta=189.6,209.6
XS Rating Curve= 0 ,0
Exp/Cntr(USF)=0,0
Exp/Cntr=0.3,0.1

Type RM Length L Ch R = 1 ,3431    ,79.7,81.8,82.7
BEGIN DESCRIPTION:
Structure 5 XS 4
END DESCRIPTION:
XS GIS Cut Line= 4
1700813.76931268 425362.452645161700833.56739068425352.192653353
1701209.82085019425279.8913233831701369.44595131 425275.06751874
#Sta/Elev= 30
       0 1082.51    16.2 1073.44    37.1 1068.86   114.5 1066.63   122.6 1065.31
   133.5 1062.24     143 1061.09   171.5 1061.51     200 1060.55   208.2 1059.49
   216.3 1055.22   220.4 1053.39   224.5 1053.02   232.4 1055.27   240.8 1057.54
   256.5 1058.72     310 1059.03   389.8  1060.8   403.7 1062.17   411.7 1064.34
   427.7 1065.32   447.7 1065.11   451.8 1066.71   459.8 1073.96   471.8 1081.09
   479.8 1086.86   483.8 1088.86   491.8 1090.51     543  1117.7   565.1 1127.37
#Mann= 5 ,-1,0
       0      .1       0   216.3    .045       0   232.4      .1       0
   312.3     .06       0  515.44      .1       0
Bank Sta=216.3,232.4
XS Rating Curve= 0 ,0
Exp/Cntr(USF)=0,0
Exp/Cntr=0.3,0.1

Type RM Length L Ch R = 1 ,3350    ,33.6,33.4,33.2
BEGIN DESCRIPTION:
Structure 5 XS 3
END DESCRIPTION:
XS GIS Cut Line= 3
1700832.33900001425392.2634362431701194.94409969425394.724556829
1701368.04291425425468.558174412
#Sta/Elev= 30
       0 1084.56     7.8 1079.52    19.8 1073.31    27.8 1070.17    35.8 1068.06
    63.8 1065.94    87.8 1065.25   119.8 1058.18   159.8 1058.07   195.8 1056.84
   206.7 1053.91   215.8 1052.66   219.8 1053.08   221.91054.062   227.8 1056.13
   239.8 1057.68   271.8 1059.44   287.8 1061.02   323.8 1062.11   364.9 1064.75
   383.2 1064.79   397.8 1066.73   446.5  1069.1     490 1072.98   507.4 1072.61
   520.4 1074.96   533.5 1074.41   537.8 1075.18   546.5 1078.83   550.8 1079.82
#Mann= 7 ,-1,0
       0      .1       0   206.7    .045       0   221.9      .1       0
     290     .07       0  382.61      .1       0  392.61     .06       0
  492.61      .1       0
Bank Sta=206.7,221.9
XS Rating Curve= 0 ,0
Exp/Cntr(USF)=0,0
Exp/Cntr=0.3,0.1

Type RM Length L Ch R = 1 ,3316    ,114.9,123.9,127.5
BEGIN DESCRIPTION:
Structure 5 XS 2
END DESCRIPTION:
XS GIS Cut Line= 3
1700831.51862648425430.0006185631701183.45887029425425.078377391
1701357.37805837425492.349006744
#Sta/Elev= 30
       0 1087.78    16.6 1078.27    24.6 1073.01    28.6  1070.9    32.6 1069.62
    48.6 1066.61    72.6 1065.24    76.6 1064.41    88.6  1059.8    96.6 1057.59
   165.5 1056.65   192.6 1057.08   204.6 1053.67   216.6 1052.41  221.961053.616
   228.6 1056.64   248.6 1058.02   324.6 1061.81   348.6 1064.16   370.6  1064.3
     387 1066.08   429.9 1067.34   454.1 1072.83   472.7 1074.39   477.1 1076.36
   481.3 1077.43   498.5 1077.89   507.1 1079.01   524.2 1084.34   538.5  1087.6
#Mann= 6 ,-1,0
       0      .1       0      90     .05       0     190     .06       0
   204.6    .045       0  221.96     .06       0  491.97      .1       0
Bank Sta=204.6,221.96
XS Rating Curve= 0 ,0
Exp/Cntr(USF)=0,0
Exp/Cntr=0.3,0.1

Type RM Length L Ch R = 1 ,3192    ,97.8,94.2,90.9
BEGIN DESCRIPTION:
Structure 4 XS 5 AND Structure 5 XS 1
END DESCRIPTION:
XS GIS Cut Line= 4
 1700809.3685412425466.0970538261700951.29316167425502.193489089
1700977.54511459425524.3435743641701296.67041725 425621.14765075
#Sta/Elev= 30
       0  1095.5    15.2 1087.68    44.1 1070.88    56.5 1066.97    81.3 1062.36
    96.4 1057.03   118.4 1056.13   143.2 1056.81   152.8 1055.56  161.181052.067
   168.5 1050.91   174.2 1052.02   179.9 1055.05     183 1055.65   195.8 1054.72
   250.4 1055.81   279.2 1057.47   311.3 1061.73   330.5 1060.91   356.2  1061.4
     359 1062.03   367.4 1066.42   384.1 1067.91   392.5 1071.39   413.4 1077.93
   421.7  1083.1   442.4 1088.64   459.4 1096.53   484.6 1111.73   514.3 1127.89
#Mann= 8 ,-1,0
       0      .1       0     120     .05       0  156.44      .1       0
  161.18    .045       0   174.2      .1       0  220.79     .05       0
  330.79     .08       0  430.79      .1       0
Bank Sta=161.18,174.2
XS Rating Curve= 0 ,0
Exp/Cntr(USF)=0,0
Exp/Cntr=0.3,0.1

Type RM Length L Ch R = 1 ,3098    ,39.4,39.4,39.1
BEGIN DESCRIPTION:
Structure 4 XS 3
END DESCRIPTION:
XS GIS Cut Line= 3
1700719.94782658425530.9065625931701134.38649996425653.233367312
1701227.36216655425738.916824754
#Sta/Elev= 30
       0 1138.64    20.8 1132.06    25.2 1130.01    36.9 1121.98    46.5 1113.89
    71.1 1095.33    91.9 1085.73   108.6 1074.26     117 1069.54   129.5 1064.44
   154.5 1058.09   162.8 1054.92   178.6 1052.85   183.7 1051.11     192 1050.05
   200.4 1051.19   207.5 1053.98   212.9 1054.61   304.6 1055.19   371.4 1059.88
   404.7 1061.01   420.1 1060.53   435.7 1067.93     447 1072.46   466.5 1084.12
   486.6 1094.62   510.6 1108.99   540.4 1125.48   548.9 1129.12   558.6 1131.77
#Mann= 6 ,-1,0
       0      .1       0   183.7    .045       0   200.4      .1       0
     310     .07       0     420     .06       0  512.11      .1       0
Bank Sta=183.7,200.4
XS Rating Curve= 0 ,0
Exp/Cntr(USF)=0,0
Exp/Cntr=0.3,0.1

Type RM Length L Ch R = 1 ,3059    ,197,199.5,201.4
BEGIN DESCRIPTION:
Structure 4 XS 2
END DESCRIPTION:
XS GIS Cut Line= 3
 1700709.2829707425566.1826243271701118.73489824425685.857278012
 1701208.9759864 425764.24852631
#Sta/Elev= 30
       0 1139.09    13.9 1135.15    23.8 1129.99    36.3 1121.24    48.8 1110.83
    69.6 1096.23    82.1 1090.71    94.5  1083.7   129.9 1059.31   140.5 1056.05
   161.3 1054.61  168.871051.278   175.1 1049.64   181.5    1050   186.3 1051.32
   191.2    1053   197.7 1053.85   250.8 1053.35   348.8 1057.54   371.7 1057.83
     403 1061.06   419.7 1060.56   423.9  1062.1   433.7 1071.31     449 1082.01
   479.5 1095.67     489 1102.95     523 1124.52   534.4 1129.72   546.1 1132.68
#Mann= 6 ,-1,0
       0      .1       0  168.87    .045       0   186.3      .1       0
     320     .07       0  426.58     .06       0  456.58      .1       0
Bank Sta=168.87,186.3
XS Rating Curve= 0 ,0
Exp/Cntr(USF)=0,0
Exp/Cntr=0.3,0.1

Type RM Length L Ch R = 1 ,2859    ,356.6,358,359.1
BEGIN DESCRIPTION:
Structure 4 XS 1
END DESCRIPTION:
XS GIS Cut Line= 6
1700598.68487181425690.649093566 1700742.6967229425765.927486328
 1700831.3185929 425812.254165321700899.16524199425844.993601156
1700979.39769307425883.6319753211701065.08682615425926.469159989
#Sta/Elev= 30
       0 1165.49     6.1 1161.71    15.2 1154.28    24.2 1149.39    87.5 1131.92
   109.9 1129.31   116.3 1127.33     125 1123.31   132.5 1117.76   159.6 1093.94
   177.6 1083.84   191.2 1070.41   200.2 1062.77   213.7 1052.07   218.3 1050.02
   230.7 1048.29   236.3 1048.72  240.181050.111   245.3 1051.71     290    1052
   352.2 1054.98     370 1055.07   419.1 1060.01   441.1 1059.89   445.6 1063.08
   451.9 1069.18   463.9 1076.26   481.3 1089.45   500.5  1102.5   522.7 1120.67
#Mann= 7 ,-1,0
       0      .1       0   218.3    .045       0  240.18      .1       0
   252.5     .06       0  367.83     .07       0  466.88     .06       0
  476.88      .1       0
Bank Sta=218.3,240.18
XS Rating Curve= 0 ,0
Exp/Cntr(USF)=0,0
Exp/Cntr=0.3,0.1

Type RM Length L Ch R = 1 ,2501    ,560.5,559.6,558.6
XS GIS Cut Line= 6
1700334.32820167425924.4289609191700414.17121784425973.563377082
1700637.73146626426111.1392174211700701.60568234 426150.44622542
1700776.12554643426196.3050575851700855.96823451426245.439801842
#Sta/Elev= 30
       0 1169.78    20.9    1163    67.9 1146.05    81.9 1139.99   124.2 1132.85
     130 1131.47   138.3 1128.22   152.6 1121.78   184.5 1102.79   196.2 1098.33
   204.9  1094.1   231.1 1085.68   255.7 1075.53   263.1 1070.04   274.5 1058.52
   280.5 1053.54   293.3 1047.05   298.2 1045.89   305.5 1045.52  311.611045.908
   321.5 1049.23   438.9 1050.19   448.3 1050.89   471.8 1054.57   501.5 1055.19
   504.4 1056.17   518.7 1070.03   542.4  1084.7   556.3  1092.3   612.5 1118.54
#Mann= 6 ,-1,0
       0      .1       0   298.2    .045       0  311.61      .1       0
  346.25     .05       0  461.25     .06       0  578.75      .1       0
Bank Sta=298.2,311.61
XS Rating Curve= 0 ,0
Exp/Cntr(USF)=0,0
Exp/Cntr=0.3,0.1

Type RM Length L Ch R = 1 ,1942    ,263.9,270.4,270.8
BEGIN DESCRIPTION:
Structure 3 XS 4
END DESCRIPTION:
XS GIS Cut Line= 6
1700108.01630073 426486.396749441700195.36848823 426520.57876769
1700276.03761824426554.479618522 1700436.7918899426623.639913264
1700486.18131376 426644.96840911 1700684.0098994426695.494100261
#Sta/Elev= 30
       0 1165.55    29.5 1149.64    51.1 1140.15    81.7  1132.3    91.3 1128.34
   129.3 1101.33   155.6 1086.19   168.4 1082.73   190.1    1067   198.8 1062.69
   216.2 1051.05   224.9 1046.31     238 1043.92   256.3 1042.46   265.1 1041.65
  269.521042.462   277.2 1045.15   356.5 1044.06   380.8 1047.32   403.5 1047.31
   407.9 1048.46   416.2 1055.16   424.5 1064.41   432.7 1072.28   440.9 1077.92
   478.2 1098.03   544.2 1136.57   556.6 1142.45   588.9 1152.28   614.3 1164.87
#Mann= 5 ,-1,0
       0      .1       0  241.31     .07       0   256.3    .045       0
  269.52     .06       0   450.1      .1       0
Bank Sta=256.3,269.52
XS Rating Curve= 0 ,0
Exp/Cntr(USF)=0,0
Exp/Cntr=0.3,0.1

Type RM Length L Ch R = 1 ,1671    ,35.6,34.5,33.9
BEGIN DESCRIPTION:
Structure 3 XS 3
END DESCRIPTION:
XS GIS Cut Line= 6
1700095.29542661426623.3537668451700192.82872392426732.736904005
1700259.37013235426765.5518451531700344.14206365426817.508835304
1700417.97568124426851.2353025941700667.73384442426868.554299311
#Sta/Elev= 30
       0 1127.89    13.3  1121.5    25.3  1114.5    49.8 1096.83    71.3 1090.36
   119.5 1060.05   134.6 1053.06   145.9 1049.45   226.5 1045.71   315.4 1044.44
   320.1  1043.5  326.12 1040.84   338.3 1039.08   343.6 1039.27  347.69 1040.81
   350.9 1042.93   355.3 1044.31   377.3 1044.02   381.7 1045.76   390.5 1054.83
   394.9 1058.19   427.1 1077.67   439.6 1086.85   459.6 1096.38   483.7 1111.65
   527.8 1134.16   583.9 1152.83     607 1166.95     632 1179.95   651.7 1188.94
#Mann= 5 ,-1,0
       0      .1       0  300.74     .06       0  326.12    .045       0
  347.69     .06       0  511.34      .1       0
Bank Sta=326.12,347.69
XS Rating Curve= 0 ,0
Exp/Cntr(USF)=0,0
Exp/Cntr=0.3,0.1

Type RM Length L Ch R = 1 ,1637    ,298,295.9,292.7
BEGIN DESCRIPTION:
Structure 3 XS 2
END DESCRIPTION:
XS GIS Cut Line= 6
 1700071.5957469426634.2920805611700178.24430563426765.551845153
1700289.45049507426813.8627307321700339.54108987426854.048162889
1700415.24110281426882.1838483881700666.82231827426894.988557458
#Sta/Elev= 30
       0 1127.08    19.9 1117.76    53.1 1097.91      75 1090.21    87.3 1084.06
     106 1072.52   127.1 1057.91     142 1050.33   175.4 1047.56   183.9  1048.2
   204.1 1046.85   294.8 1045.92   311.4 1044.52   320.4 1044.84   345.3 1043.36
  356.131039.728   366.5 1038.86   372.5 1039.76     381 1043.59   410.9 1043.31
   415.1 1045.68   419.4 1050.53   440.4 1069.83   460.5 1082.61   480.5 1091.31
   507.2 1106.83   552.6  1131.1   604.6 1148.61   664.7 1179.75   687.5 1189.38
#Mann= 5 ,-1,0
       0      .1       0  340.58     .06       0  356.13    .045       0
   372.5     .06       0  445.55      .1       0
Bank Sta=356.13,372.5
XS Rating Curve= 0 ,0
Exp/Cntr(USF)=0,0
Exp/Cntr=0.3,0.1

Type RM Length L Ch R = 1 ,1341    ,337.1,337.5,337.2
BEGIN DESCRIPTION:
Structure 3 XS 1
END DESCRIPTION:
XS GIS Cut Line= 2
1700025.77083164427150.2047908441700645.42850715427149.426772422
#Sta/Elev= 30
       0 1122.46    22.3  1112.2    54.3 1092.56    68.8 1087.55    86.3 1079.83
   110.3 1066.86   122.3 1058.95   138.3 1050.01   146.3 1046.69   170.3 1043.26
   302.3 1039.37  309.571037.048   314.3 1036.12   326.3 1036.95   334.3 1040.36
   350.3 1040.92   354.3  1041.9   362.3 1053.62   366.3 1056.72   398.3 1070.76
   414.3 1080.93   418.3 1081.92   434.3 1082.58   446.3 1091.44   465.3  1102.9
   494.3 1123.16   502.3 1127.53   570.3 1149.56   594.3 1165.79   619.7 1178.46
#Mann= 4 ,-1,0
       0      .1       0  309.57    .045       0   326.3     .06       0
     400      .1       0
Bank Sta=309.57,326.3
XS Rating Curve= 0 ,0
Exp/Cntr(USF)=0,0
Exp/Cntr=0.3,0.1

Type RM Length L Ch R = 1 ,1003    ,147.1,144.7,145.1
BEGIN DESCRIPTION:
Structure 2 XS 4
END DESCRIPTION:
XS GIS Cut Line= 6
1700027.37212268427476.1086003331700121.99496493427478.926508084
1700210.48822625427482.2050448361700286.33518742427485.197821006
  1700386.514449427485.3119940011700642.53296584427474.420939669
#Sta/Elev= 30
       0 1150.31    24.8 1141.33    56.8 1131.93    68.8 1125.29    80.8 1121.01
   124.8 1091.37   152.8 1081.59   184.8 1063.11   216.9 1039.89   236.9 1037.28
   292.9 1037.69  303.551034.255   308.9 1033.33   316.9 1034.31   328.9 1038.61
   348.9 1038.86   352.9 1040.25   356.9 1043.29   364.9 1055.93   368.9 1060.53
   384.9 1072.63   400.9 1080.36     433 1090.39     485 1126.74     505 1137.05
     513 1139.18   525.1  1139.6   549.1 1150.65   595.8 1182.04   615.6 1193.54
#Mann= 4 ,-1,0
       0      .1       0  303.55    .045       0   316.9     .06       0
   399.3      .1       0
Bank Sta=303.55,316.9
XS Rating Curve= 0 ,0
Exp/Cntr(USF)=0,0
Exp/Cntr=0.3,0.1
